--- sprngfrk.prj (project) ---

Proj Title=sprngfrk
Current Plan=p01
Default Exp/Contr=0,0
English Units
Geom File=g01
Flow File=f01
Plan File=p01
BEGIN DESCRIPTION:
END DESCRIPTION:
DSS Export Rating Curves= 0
DSS Export Rating Curve Sorted= 0
DSS Export Volume Flow Curves= 0
DXF OffsetX= 0
DXF OffsetY= 0
DXF ScaleX= 0
DXF ScaleY= 0

--- sprngfrk.p01 (plan) ---

Plan Title=Floodplain
Program Version=4.00
Geom File=g01
Flow File=f01
K Sum by GR=0
Std Step Tol=0.01
Critical Tol=0.01
Num of Std Step Trials=20
Max Error Tol=0.3
Flow Tol Ratio=0.001
Split Flow NTrial=30
Split Flow Tol=0.02
Split Flow Ratio=0.02
Log Output Level=0
Friction Slope Method=1
Unsteady Friction Slope Method=2
Unsteady Bridges Friction Slope Method=1
Global Log Level=0
CheckData=False
Run HTab=0
Run UNet=0
Run PostProcess=0
UNET Theta=0
UNET Theta Warmup=0
UNET ZTol=0
UNET ZSATol=0
UNET MxIter=0
UNET MaxInSteps=0
UNET DtIC=0
UNET DtMin=0
UNET MaxCRTS=0
UNET WFStab=0
UNET SFStab=0
UNET WFX=0
UNET SFX=0
UNET DSS MLevel=0
UNET DZMax Abort=0
UNET Convert EG Bridges=0
UNET Use Existing IB Tables=0
UNET Froude Limit=0
UNET Froude Power=0
Write IC File=0
Echo Input=False
Echo Output=False
Write Detailed=0

--- sprngfrk.f01 (steady flow) ---

Flow Title=NFF Regression Equation
Program Version=4.00
Number of Profiles= 1
Profile Names=P100yr
River Rch & RM=sprngfrk,Main            ,13204.7
     306
River Rch & RM=sprngfrk,Main            ,12730.4
     363
River Rch & RM=sprngfrk,Main            ,12488.4
     374
River Rch & RM=sprngfrk,Main            ,11234.6
     412
River Rch & RM=sprngfrk,Main            ,9944.2
     445
River Rch & RM=sprngfrk,Main            ,8838.7
     481
River Rch & RM=sprngfrk,Main            ,7914.9
     517
River Rch & RM=sprngfrk,Main            ,7705.6
     573
River Rch & RM=sprngfrk,Main            ,4391.3
     629
River Rch & RM=sprngfrk,Main            ,4095.2
     962
River Rch & RM=sprngfrk,Main            ,287.3
    1017
Boundary for River Rch & Prof#=sprngfrk,Main            , 1
Up Type= 0
Dn Type= 3
Dn Slope=0.026
DSS Import GetInterval= 0
DSS Import GetPeak= 0
DSS Import FillOption= 0

--- sprngfrk.g01 (geometry) ---

Geom Title=USGS 10m DEM
Program Version=4.00

River Reach=sprngfrk        ,Main
Reach XY= 30
     1702293.351      203077.662     1702266.034      203136.108
      1702134.03      203140.286     1701657.577      203377.167
     1701352.293      203598.924     1701235.614       203804.89
     1700774.798      203897.138     1700020.767      203617.508
     1699786.861      203442.695     1699656.668       203253.72
     1699283.455      203107.667     1699056.388      202926.673
     1698920.738      202950.132     1698335.779      202790.149
     1697442.623      202946.874     1696742.258      203419.233
     1696482.363      203694.428     1696231.818       203798.24
     1696066.703       204049.77     1695830.129      204131.468
     1695672.677      204333.171     1695533.558      204970.917
     1695206.823      205494.524     1695012.646      205513.616
     1694632.368      205721.161     1694073.607      205873.363
     1692798.398      206628.205     1692602.317      206676.197
     1692443.944      206814.687     1691582.641      206923.219

Type RM Length L Ch R = 1 ,13204.7 ,232.4,248.3,264.2
XS GIS Cut Line= 4
     1701890.586      202752.461     1702234.907      203069.813
     1702371.341      203095.865     1702707.283      203115.176
#Sta/Elev= 30
      10 1430.74    29.9 1415.03    79.7 1382.67    89.7 1377.05    99.6 1375.28
   119.6 1364.18   139.5 1351.18   159.4 1335.19   209.2 1303.06   249.1 1279.04
   358.7 1219.77   378.6 1206.12   418.4 1189.58   478.2 1179.74   517.8 1175.75
   527.8  1175.6   537.8 1177.25   547.6 1180.87   567.5 1193.19     627 1216.29
   636.9 1224.29   706.1 1261.83     716 1271.49   775.4 1299.71   785.3 1308.05
   795.2 1313.58   854.6 1341.96   874.4 1354.51     914 1370.08   943.7 1385.52
#Mann= 3 , 0 , 0
       0      .1       0   517.8    .045       0   537.8      .1       0
Bank Sta=517.8,537.8
XS Rating Curve= 0 ,0
Exp/Cntr=0.3,0.1

Type RM Length L Ch R = 1 ,12956.4 ,222.4,226,229.6
XS GIS Cut Line= 4
     1701882.739      202758.666     1702023.515      203068.556
     1702129.554      203218.473     1702131.382      203509.166
#Sta/Elev= 30
      10  1427.1      40 1404.11    50.1 1398.21    60.1 1396.37    70.1 1388.95
   100.1 1363.97   110.1    1357   170.2 1317.88   180.2 1316.58   240.3 1274.29
   290.3 1241.44   300.3 1238.02   330.4 1221.11     408 1181.96   427.3  1177.6
     437 1173.92     456 1170.56     466 1169.03     476 1170.06     495 1175.26
     544 1186.21   554.1 1186.32   604.2 1198.63   614.2 1202.98   644.3 1220.43
   654.3 1220.72   744.5 1271.44   754.5 1272.39   764.6 1277.35   814.7 1305.99
#Mann= 3 , 0 , 0
       0      .1       0     456    .045       0     476      .1       0
Bank Sta=456,476
XS Rating Curve= 0 ,0
Exp/Cntr=0.3,0.1

Type RM Length L Ch R = 1 ,12730.4 ,96.7,95.1,93.5
XS GIS Cut Line= 4
     1701854.401      202764.151     1701851.659      203177.337
     1701927.531      203339.138     1702080.191      203528.362
#Sta/Elev= 30
    10.1 1427.27    30.2 1411.94    40.3 1406.27    50.4 1404.57     131 1344.23
   141.1 1338.17   151.2 1336.89   211.6 1293.63   241.9  1275.3   251.9 1274.52
   282.2 1255.36   312.4 1241.21   342.6 1223.81   352.7 1223.48   413.2 1190.39
   452.9 1170.68   492.5 1162.51   502.5 1161.05   512.5 1162.26   562.1 1183.21
     572 1186.42     582 1187.42   622.3  1203.8   652.7  1220.7   703.3 1251.57
   713.5  1255.8   723.6 1257.78     754  1275.8   794.5 1298.57     835 1318.62
#Mann= 3 , 0 , 0
       0      .1       0   492.5    .045       0   512.5      .1       0
Bank Sta=492.5,512.5
XS Rating Curve= 0 ,0
Exp/Cntr=0.3,0.1

Type RM Length L Ch R = 1 ,12635.3 ,149.2,146.9,144.6
XS GIS Cut Line= 4
     1701760.246      202797.059     1701747.448      203201.104
      1701845.26      203372.046     1701965.925       203552.13
#Sta/Elev= 30
    10.1 1402.19    50.5 1374.78      91 1349.67   111.2 1342.28   151.6 1311.31
   171.8 1298.85     192  1289.5   212.2 1285.31   242.5 1271.72   293.1 1239.47
   313.3 1232.97   333.5 1220.62     384 1195.17   404.2 1186.18   414.1  1183.3
   423.9  1182.8   473.2 1168.21   492.9 1164.65  505.83 1160.98   512.6 1159.25
  528.11 1160.72   542.1 1163.71   561.8 1173.24   630.8 1202.41   660.3 1217.05
   670.2 1218.51   689.9  1229.6   788.4 1289.45   808.1    1296     818    1302
#Mann= 3 , 0 , 0
    10.1      .1       0  505.83    .045       0  528.11      .1       0
Bank Sta=505.83,528.11
XS Rating Curve= 0 ,0
Exp/Cntr=0.3,0.1

Type RM Length L Ch R = 1 ,12488.4 ,205.8,203.7,201.6
XS GIS Cut Line= 4
     1701366.256        203058.5     1701617.642      203291.603
     1701716.368       203425.98     1701915.648      203587.781
#Sta/Elev= 30
    10.1 1358.48    40.3 1344.87    50.4 1336.61    60.5  1330.8    90.7 1315.96
   110.9 1307.28   161.3 1287.86   181.5 1277.41   191.6 1274.31   211.7 1262.38
     242 1239.71   272.2 1222.49   292.4  1209.6   352.6 1182.42   362.4 1181.15
   401.7 1163.45  427.76 1155.72   440.9 1154.55  447.69 1156.49     490 1174.48
   499.8 1175.58   519.4 1182.27   539.2 1191.18   588.6 1210.95   647.8 1242.17
   657.7 1249.46   677.4 1254.89   697.2 1265.43   746.5 1293.12   766.3 1307.14
#Mann= 3 , 0 , 0
    10.1      .1       0  427.76    .045       0  447.69      .1       0
Bank Sta=427.76,447.69
XS Rating Curve= 0 ,0
Exp/Cntr=0.3,0.1

Type RM Length L Ch R = 1 ,12284.7 ,183.9,183.3,182.8
XS GIS Cut Line= 4
     1701283.985      203121.727     1701452.185      203425.218
     1701554.567      203537.351     1701795.897      203688.487
#Sta/Elev= 30
     9.9 1376.12    29.7    1360    49.6 1347.36    59.5 1345.22    69.4 1341.25
   128.9 1305.37   158.6 1288.48   168.5 1283.22   178.4 1281.87   247.8 1238.29
   287.5 1214.84   297.4 1209.54   307.3 1206.41   317.2 1199.83   387.5 1162.26
   407.7 1153.13     418 1149.98     428 1147.98     438 1148.55   448.2 1149.92
   488.7 1161.72   538.1 1179.04   557.7 1189.66   616.7 1216.61   636.3 1227.25
   646.1 1234.11   665.7 1241.38   724.7 1273.09   744.3 1287.01   783.6 1308.01
#Mann= 3 , 0 , 0
       0      .1       0     418    .045       0     438      .1       0
Bank Sta=418,438
XS Rating Curve= 0 ,0
Exp/Cntr=0.3,0.1

Type RM Length L Ch R = 1 ,12101.4 ,327.6,339.7,351.8
XS GIS Cut Line= 4
     1701029.248      203335.024     1701305.924      203537.351
     1701439.996      203676.299     1701695.952      203785.994
#Sta/Elev= 30
    10.1 1366.69    20.2 1357.79    30.2 1350.74    40.3 1347.66    80.6 1323.45
   110.9  1308.2   131.1 1294.47   141.1  1288.9   211.7  1250.7     252 1230.51
   292.4 1204.59   312.5 1193.17   332.7 1180.21     391 1154.08   400.7  1148.8
   410.3 1145.49   419.6  1144.4   429.7 1143.49   439.6 1144.81   477.9 1149.86
   535.8 1168.37   555.7 1176.74   575.6 1183.46   615.4 1195.28   635.3 1204.89
   645.2 1211.53   714.9 1243.62   734.8 1256.37   804.4 1290.26   814.3 1297.86
#Mann= 3 , 0 , 0
       0      .1       0   419.6    .045       0   439.6      .1       0
Bank Sta=419.6,439.6
XS Rating Curve= 0 ,0
Exp/Cntr=0.3,0.1

Type RM Length L Ch R = 1 ,11761.7 ,134.1,128.9,123.6
XS GIS Cut Line= 4
     1700997.558      203353.307     1701134.068      203715.302
     1701166.976      203896.909     1701255.952      204135.801
#Sta/Elev= 30
     9.9 1377.14    59.5 1341.07    99.2 1310.33     119 1302.61     129 1295.99
   158.7 1278.43   178.6 1265.31   208.3 1248.19   228.2 1242.23   287.7  1208.3
   327.4 1186.61   347.2  1180.8   386.9 1162.35   435.4 1143.55   445.2 1142.77
   464.6 1138.61   483.7  1136.8   493.7  1136.6   503.7 1137.74   522.9 1142.94
     552 1152.35   561.7 1153.01   591.1 1163.71   600.9 1167.83   649.9 1195.34
   659.7 1200.24   669.5 1201.23   777.3 1270.99   787.1 1271.55   826.4  1295.1
#Mann= 3 , 0 , 0
       0      .1       0   483.7    .045       0   503.7      .1       0
Bank Sta=483.7,503.7
XS Rating Curve= 0 ,0
Exp/Cntr=0.3,0.1

Type RM Length L Ch R = 1 ,11632.8 ,113.9,121.4,129
XS GIS Cut Line= 4
     1700956.117      203367.933     1700980.494      203740.897
     1701073.126      203932.255     1701199.885      204129.707
#Sta/Elev= 30
    10.1 1385.34    30.3 1370.13    70.7 1336.84    80.8 1334.96   121.2 1308.06
   171.7 1280.86   181.8 1279.35   191.9 1275.47   282.8 1226.23   292.9 1224.08
     303 1219.56   383.9  1166.9   404.1 1160.17   424.4 1148.09   434.5 1144.62
   464.9 1139.24   485.2 1134.33   495.2 1132.93   505.2 1133.19   525.6  1134.6
   535.7 1137.07   605.9 1165.54   615.7 1170.08   625.5 1175.95     645  1182.4
   752.6 1246.03   762.3 1251.25   772.1 1252.13   781.9 1257.55     821 1282.31
#Mann= 3 , 0 , 0
       0      .1       0   485.2    .045       0   505.2      .1       0
Bank Sta=485.2,505.2
XS Rating Curve= 0 ,0
Exp/Cntr=0.3,0.1

Type RM Length L Ch R = 1 ,11511.4 ,145.8,149.6,153.5
XS GIS Cut Line= 4
     1700907.364      203416.686     1700912.239      203783.556
     1700928.084      203987.102     1701032.904      204183.336
#Sta/Elev= 30
     9.9 1357.75    19.8  1349.8    39.7 1341.62    59.5 1326.78     119 1295.56
   128.9 1292.17   138.8 1290.99   148.7 1286.96   228.1 1242.97     238 1242.02
   297.5 1194.21   327.2 1174.95   337.2 1174.48   366.9 1160.85   405.8 1146.43
   425.2 1139.69   444.7 1136.39   463.8 1129.26   473.8 1127.83   483.8 1128.26
   522.5 1132.82   541.9  1139.9   551.6 1140.02   591.3 1156.32     652 1198.62
   662.1 1200.28   672.2 1206.04   712.6 1232.51   773.3 1269.68   793.5 1276.77
#Mann= 3 , 0 , 0
       0      .1       0   463.8    .045       0   483.8      .1       0
Bank Sta=463.8,483.8
XS Rating Curve= 0 ,0
Exp/Cntr=0.3,0.1

Type RM Length L Ch R = 1 ,11361.8 ,124.6,127.2,129.8
XS GIS Cut Line= 4
     1700853.735       203402.06     1700779.386      203824.997
     1700757.447      204017.574     1700886.643      204235.746
#Sta/Elev= 30
      10 1383.68      30 1361.34    39.9 1360.78    49.9 1352.47    69.9 1342.16
   109.9 1329.61   129.8 1321.43   139.8 1321.23   159.8 1312.71   209.7 1285.92
   229.7 1273.44   249.7 1266.88   329.6 1211.68   339.5 1206.39   349.5 1205.66
   399.5 1173.32   439.1 1150.52   448.8 1149.76   458.5 1145.44   487.6 1127.75
     497  1123.8     507  1122.9     517 1124.44   555.4 1128.54     672 1151.98
   740.3 1177.64   779.3  1195.3     789 1196.98   818.3 1215.25   876.8 1245.99
#Mann= 3 , 0 , 0
       0      .1       0     497    .045       0     517      .1       0
Bank Sta=497,517
XS Rating Curve= 0 ,0
Exp/Cntr=0.3,0.1

Type RM Length L Ch R = 1 ,11234.6 ,262.5,266.4,270.2
XS GIS Cut Line= 4
     1700772.073      203408.154     1700673.347      203765.274
     1700625.812       203957.85     1700411.297       204189.43
#Sta/Elev= 30
      10 1397.59      20 1396.12    50.1 1376.88    90.1 1360.92   110.2 1350.04
   120.2 1345.65   130.2 1344.71   220.3 1285.49   240.3 1278.92   320.4 1220.93
   330.5 1215.14   340.5 1213.59   390.4 1177.21     430 1143.94   439.9 1141.31
   459.8 1125.29   469.6  1120.2   479.6 1119.64   489.6 1120.88   539.1  1126.6
   618.2 1130.79   677.4 1140.94     707 1148.91   726.7 1157.25   746.4 1168.68
   766.2 1185.66   785.9 1199.16   805.6 1207.19   864.8 1251.34   884.5 1263.04
#Mann= 3 , 0 , 0
       0      .1       0   469.6    .045       0   489.6      .1       0
Bank Sta=469.6,489.6
XS Rating Curve= 0 ,0
Exp/Cntr=0.3,0.1

Type RM Length L Ch R = 1 ,10968.2 ,195.4,199.4,203.4
XS GIS Cut Line= 4
     1700656.283      203382.559     1700445.424       203675.08
     1700372.294      203833.529        1700198.      204082.172
#Sta/Elev= 30
      10 1404.05      30 1394.03    50.1 1388.29    80.1 1372.24    90.1 1366.27
   110.2 1350.79   150.2 1324.91   160.3 1319.01   170.3 1317.04   190.3 1304.81
   210.3 1291.44   230.4 1274.75   270.4 1246.55   280.5 1243.91   300.5 1231.46
   330.5 1209.84   350.6 1191.72   389.7 1162.86   409.1 1153.58   447.9 1117.35
   457.2 1114.63   457.5 1114.54   477.2 1115.31   525.4 1117.58   575.6 1122.87
   616.1 1133.57   626.2 1134.91   666.7 1151.18   707.2 1164.86   838.8 1225.83
#Mann= 3 , 0 , 0
       0      .1       0   457.2    .045       0   477.2      .1       0
Bank Sta=457.2,477.2
XS Rating Curve= 0 ,0
Exp/Cntr=0.3,0.1

Type RM Length L Ch R = 1 ,10768.8 ,136,128.2,120.4
XS GIS Cut Line= 4
     1700551.463      203327.711     1700290.632      203589.761
     1700169.967      203754.304     1699970.077      203931.036
#Sta/Elev= 30
      10 1379.06      50 1357.82    69.9 1343.83    99.9 1328.54   119.9 1321.38
   139.9 1310.16   149.9 1304.52   169.9 1289.22   189.9 1278.05   229.8 1256.89
   249.8 1250.11   269.8 1235.06   359.7 1179.16   379.5 1169.66   447.5 1127.03
   466.9 1110.38  469.27 1109.77   476.6 1107.96   486.6 1108.79   525.2 1110.55
   564.1 1118.88   573.8 1122.31   603.4 1137.28   623.2 1141.94   662.7 1159.49
   702.2  1182.2   751.7 1213.52   771.4 1223.12   781.3 1230.82   840.6 1269.25
#Mann= 3 , 0 , 0
      10      .1       0  469.27    .045       0   486.6      .1       0
Bank Sta=469.27,486.6
XS Rating Curve= 0 ,0
Exp/Cntr=0.3,0.1

Type RM Length L Ch R = 1 ,10640.6 ,244.6,241.5,241.6
XS GIS Cut Line= 4
     1700505.147      203306.991     1700133.402      203547.102
     1700098.055      203688.487     1699957.889      203912.754
#Sta/Elev= 30
    10.1 1366.95    70.4 1336.03    90.5 1321.98   150.9 1289.93     171 1283.78
     181 1275.81   251.4 1242.29   271.6 1227.17   321.9 1195.33     342 1186.48
     352 1176.38   372.1 1164.58   422.4 1143.41     462 1123.83   481.4 1118.48
   500.8 1108.84   510.3 1105.99   520.3 1104.28   530.3 1104.72   588.3  1119.8
   617.7 1132.67   666.6 1162.43   686.2 1170.19   705.8  1174.1   725.4 1181.33
     745 1194.83   764.6 1211.15     794 1230.96   813.6 1238.53   852.7 1264.51
#Mann= 3 , 0 , 0
       0      .1       0   510.3    .045       0   530.3      .1       0
Bank Sta=510.3,530.3
XS Rating Curve= 0 ,0
Exp/Cntr=0.3,0.1

Type RM Length L Ch R = 1 ,10399.2 ,153.1,166.6,180
XS GIS Cut Line= 4
     1700340.604      203169.262     1699939.606      203436.188
     1699900.603      203588.543     1699837.224      203857.906
#Sta/Elev= 30
      10 1365.36    70.2 1339.88    80.3 1334.09   100.4 1316.83   110.4 1310.66
   150.5 1286.71   170.6 1277.39   180.6 1267.91   250.9 1228.76     271 1212.98
   331.2 1179.86   351.2 1167.22   361.3 1164.01   441.6 1124.88   481.7 1109.61
   560.2 1100.13   570.2 1098.65   580.2 1100.86   599.7 1115.48   609.5 1117.08
   619.3 1121.52   698.3 1164.17   708.2 1168.15     718 1169.68   747.7 1185.62
   787.2 1212.09     807 1227.05   816.9 1230.45   826.8 1236.04   915.7 1296.37
#Mann= 3 , 0 , 0
       0      .1       0   560.2    .045       0   580.2      .1       0
Bank Sta=560.2,580.2
XS Rating Curve= 0 ,0
Exp/Cntr=0.3,0.1

Type RM Length L Ch R = 1 ,10232.6 ,298.3,288.4,278.4
XS GIS Cut Line= 4
     1699942.044       202962.06     1699856.725      203378.902
     1699731.185       203475.19     1699682.431      203770.149
#Sta/Elev= 30
    10.1 1305.45    40.5 1287.37    70.9 1266.11    91.2 1258.95   172.2 1208.22
   192.5 1202.47   243.1 1174.97   273.5 1160.45   283.7 1156.78   293.8 1155.71
   354.6 1129.56     385 1119.09   395.1 1118.71   425.5 1108.83     465 1099.69
   504.5 1094.17   514.5 1093.04   524.5 1093.55   534.3 1094.26   544.1  1097.2
     554 1103.69   593.7    1119   633.5 1143.59   643.5 1148.04   653.5 1149.25
   743.1 1199.48   753.1 1200.03   842.8  1256.9   862.7 1262.98   882.7 1275.28
#Mann= 3 , 0 , 0
       0      .1       0   504.5    .045       0   524.5      .1       0
Bank Sta=504.5,524.5
XS Rating Curve= 0 ,0
Exp/Cntr=0.3,0.1

Type RM Length L Ch R = 1 ,9944.2  ,244.5,244.2,243.9
XS GIS Cut Line= 4
     1699710.465      202929.151     1699643.429      203142.448
     1699581.268      203278.958     1699438.664      203480.066
#Sta/Elev= 30
     9.7 1243.67    38.9 1226.23    87.5 1198.59    97.2 1196.16   106.9 1192.24
   136.1 1176.78     175 1157.18   194.4 1146.49   204.1  1143.6   213.9 1138.28
   223.6  1131.5   243.6 1119.98   263.6 1109.53   293.6 1094.98   303.6 1090.73
   313.6  1089.5   323.6 1089.31   333.6 1090.18   373.6  1093.1   442.6    1096
   462.3 1097.22   472.2 1098.55   482.1 1102.17   491.9 1107.63   501.8 1112.53
   531.4 1126.04   551.1 1131.43   580.7 1146.41   600.4 1160.47   620.1 1170.79
#Mann= 3 , 0 , 0
       0      .1       0   313.6    .045       0   333.6      .1       0
Bank Sta=313.6,333.6
XS Rating Curve= 0 ,0
Exp/Cntr=0.3,0.1

Type RM Length L Ch R = 1 ,9700.1  ,259.6,266.2,272.8
XS GIS Cut Line= 4
     1699461.822      202810.924     1699419.162      203044.941
     1699342.376      203220.453      1699211.96      203469.096
#Sta/Elev= 30
     9.9 1281.01    79.3 1230.04    99.1 1223.34   138.8 1195.99   168.5 1171.08
   188.3 1157.33   198.2 1156.45   237.9 1130.47   288.3 1103.55   308.5 1098.73
   328.6 1088.65   338.8 1084.94   348.8 1084.31   358.8 1085.77   429.4 1086.48
   439.5 1087.33   449.5 1090.36   499.6 1117.96   509.7 1122.15   519.7 1123.99
   539.8    1136   559.8 1150.92   569.8 1157.04   599.9 1172.55     620 1184.63
     630 1186.32     640 1191.38   680.1    1217   700.2 1235.49   710.2 1243.03
#Mann= 3 , 0 , 0
     9.9      .1       0   338.8    .045       0   358.8      .1       0
#XS Ineff= 2 , 0
       0                     369       0
Permanent Ineff=
       F       F
Bank Sta=338.8,358.8
XS Rating Curve= 0 ,0
Exp/Cntr=0.3,0.1

Type RM Length L Ch R = 1 ,9433.9  ,160.1,144.3,128.4
XS GIS Cut Line= 4
     1699350.907      202796.298     1699203.428      202949.871
     1699082.763      203081.506     1699019.384      203354.525
#Sta/Elev= 30
     9.7 1259.27      29 1247.82    48.4 1231.04   106.5 1191.05   116.1 1188.73
   125.8  1184.1   135.5  1177.6   145.2 1168.64   164.5 1154.28   232.8 1108.54
   242.7 1104.43   262.5 1086.15   272.4 1079.32   282.4 1077.74   292.4 1077.88
     332 1078.78   341.9 1079.86   371.7 1084.87   391.5 1086.52   431.5 1094.16
   471.6 1107.91   481.6 1110.74   491.6 1111.68   521.6 1122.24   551.7 1129.82
   581.7 1141.47   591.7 1142.51   601.7 1145.97   651.8 1168.36   671.8 1178.32
#Mann= 3 , 0 , 0
       0      .1       0   272.4    .045       0   292.4     .08       0
Bank Sta=272.4,292.4
XS Rating Curve= 0 ,0
Exp/Cntr=0.3,0.1

Type RM Length L Ch R = 1 ,9289.6  ,219.9,229.9,239.9
XS GIS Cut Line= 4
     1699239.993      202714.635     1699036.447      202868.209
     1699044.979       203066.88     1699003.539        203339.9
#Sta/Elev= 30
     9.8 1214.49    19.6 1207.35    29.4 1202.79    68.6 1186.41    88.3 1179.87
    98.1 1175.17   107.9 1169.17   137.3 1156.54   176.5 1137.23   186.3 1130.33
   196.1 1122.15   225.6 1103.02   235.4 1097.95     255 1089.91   284.8 1082.21
   304.6 1075.91   314.6  1074.5   324.6 1074.65   404.1 1077.43   443.9 1084.48
   453.8 1084.73   503.1  1094.1   542.6 1111.26   552.5 1112.34     582 1122.79
   621.5  1133.6   641.2 1140.83   651.1 1143.76   660.9 1145.31     730 1177.99
#Mann= 3 , 0 , 0
       0      .1       0   304.6    .045       0   324.6     .08       0
Bank Sta=304.6,324.6
XS Rating Curve= 0 ,0
Exp/Cntr=0.3,0.1

Type RM Length L Ch R = 1 ,9059.7  ,223.4,221,218.6
XS GIS Cut Line= 4
     1698779.272      202583.001     1698870.685      202809.705
     1698770.741      203018.126     1698717.112      203304.553
#Sta/Elev= 30
     9.8 1206.66    39.1  1190.5    48.9 1189.81    58.7    1185   156.4 1127.98
   166.2 1125.89     176 1122.81   215.1 1102.65   244.4  1089.8   264.5 1083.07
   284.6 1080.47   324.8 1070.54   334.9 1068.89     345 1068.22     355 1068.14
     365 1068.45   425.3 1070.68   485.6  1071.3   505.7 1072.76   515.8  1076.9
   525.8 1083.75     566 1113.98   576.1 1120.54   596.2 1131.56   606.2 1131.69
   646.4 1153.08   696.7 1183.74   706.7 1185.38   716.7 1190.04     767 1224.31
#Mann= 3 , 0 , 0
       0      .1       0     345    .045       0     365     .08       0
Bank Sta=345,365
XS Rating Curve= 0 ,0
Exp/Cntr=0.3,0.1

Type RM Length L Ch R = 1 ,8838.7  ,241,238.8,236.5
XS GIS Cut Line= 4
      1698665.92       202584.22     1698636.668      202774.359
     1698586.696      202921.838     1698537.942      203233.861
#Sta/Elev= 30
    10.1  1206.7    20.3 1199.48    40.5 1192.21      81 1164.53   121.5 1139.76
   131.6 1135.72   141.8 1133.58   192.4  1104.6   231.3 1080.53     241 1079.53
   250.8 1073.95   260.5 1067.35     270 1064.09     280 1063.79     290 1064.67
   328.6  1067.5     358 1068.47   367.8 1069.53   417.2 1079.77     427 1082.65
   436.9 1086.43   456.7 1090.82     506  1111.9   545.5 1129.96   555.3  1130.3
   594.8 1148.32   634.3 1165.52   644.2 1169.46     654 1170.96   663.9 1173.54
#Mann= 3 , 0 , 0
       0      .1       0     270    .045       0     290     .08       0
Bank Sta=270,290
XS Rating Curve= 0 ,0
Exp/Cntr=0.3,0.1

Type RM Length L Ch R = 1 ,8599.9  ,157.3,150.6,143.8
XS GIS Cut Line= 4
     1698431.903      202550.092     1698395.338      202724.386
     1698361.211      202880.397     1698327.083       203129.04
#Sta/Elev= 30
     9.9 1195.93    19.8 1183.04    29.7  1173.3    39.6 1165.77    49.5 1165.41
    59.4 1158.78    79.2 1144.75      89 1138.22   108.8 1126.17   138.5 1109.47
   158.3 1104.25   188.1 1088.19     218 1072.79     238 1060.98   247.9 1058.49
   257.9 1058.43   267.9 1059.23   287.9 1062.51   297.9 1062.95   337.8 1062.57
   357.9 1063.58   367.9 1066.35   448.2  1107.3   468.3 1112.61   498.4 1128.61
   518.5 1138.38   548.6 1153.91   558.6 1157.61   568.7 1159.32   588.8 1169.92
#Mann= 3 , 0 , 0
       0      .1       0   247.9    .045       0   267.9      .1       0
Bank Sta=247.9,267.9
XS Rating Curve= 0 ,0
Exp/Cntr=0.3,0.1

Type RM Length L Ch R = 1 ,8449.4  ,220.9,222.2,223.6
XS GIS Cut Line= 4
     1698359.992      202550.092      1698225.92      202735.356
     1698247.859      202924.276     1698269.798      203105.882
#Sta/Elev= 30
     9.9 1179.32    29.8 1165.83    39.8 1160.78    49.7 1157.78    59.7 1150.72
    79.5 1135.58    89.5 1126.46    99.4  1118.3   109.4  1111.3   139.2 1092.68
   159.1 1079.41     169 1076.75   188.9 1068.94   198.9 1066.26   208.8 1065.14
   288.7 1060.59   318.8 1053.69   328.8  1053.4   338.8 1054.35   368.8 1059.09
   378.8 1062.12   388.8 1062.76   438.1 1089.06   476.6 1108.89   486.3 1110.39
   495.9 1113.59   524.8 1129.02   572.9 1155.61   582.5 1160.33   601.8 1165.54
#Mann= 3 , 0 , 0
       0      .1       0   318.8    .045       0   338.8      .1       0
Bank Sta=318.8,338.8
XS Rating Curve= 0 ,0
Exp/Cntr=0.3,0.1

Type RM Length L Ch R = 1 ,8227.1  ,311.8,312.2,312.5
XS GIS Cut Line= 4
     1697835.892      202470.868     1698015.061      202728.043
     1698023.593      202925.494     1698027.249      203138.791
#Sta/Elev= 30
    10.1 1212.14    20.2 1203.34    30.3 1195.67    60.7 1173.69    80.9 1160.04
      91 1157.33   101.1 1152.99   151.7 1124.66   161.8 1116.68   171.9 1107.47
   192.1 1087.45   202.2 1078.42   212.3 1073.97   232.5 1072.83   343.1 1061.17
   392.5    1057   441.8 1047.62   451.8 1047.37   461.8 1047.98   471.5 1050.54
   491.3 1060.31   511.1 1073.26   549.9  1105.6   559.6 1105.52   578.9 1121.27
   598.3 1134.79   627.4 1150.47   646.8 1162.67   666.2 1168.83   724.4 1206.34
#Mann= 3 , 0 , 0
       0      .1       0   441.8    .045       0   461.8      .1       0
Bank Sta=441.8,461.8
XS Rating Curve= 0 ,0
Exp/Cntr=0.3,0.1

Type RM Length L Ch R = 1 ,7914.9  ,209,209.4,209.8
XS GIS Cut Line= 4
      1697774.95      202467.211     1697710.351      202808.486
     1697714.008      202943.777     1697765.199      203091.256
#Sta/Elev= 30
     9.9 1213.38    39.7 1188.17    59.5 1174.09    69.5 1172.24    79.4 1168.19
     129 1138.42   158.8 1121.67   168.7 1117.86   178.6 1115.77   188.6 1108.24
   238.2 1064.78   248.1 1058.94   267.9 1056.67   277.9 1056.61   366.7  1049.4
     386 1048.69   395.7 1047.61     405 1045.65     415 1043.67     425 1044.89
     473 1071.85   482.7 1071.88   492.4 1077.68   521.7 1097.26     551 1120.02
     590 1147.78   599.8 1148.56   609.5 1152.79   619.3  1154.7   638.8 1155.98
#Mann= 3 , 0 , 0
       0     .06       0     405    .045       0     425      .1       0
Bank Sta=405,425
XS Rating Curve= 0 ,0
Exp/Cntr=0.3,0.1

Type RM Length L Ch R = 1 ,7705.6  ,213.3,198,182.6
XS GIS Cut Line= 4
     1697248.412      202721.948     1697521.628      202904.948
     1697522.997      203021.289     1697607.553       203151.52
#Sta/Elev= 30
       0 1137.28      10 1137.28    19.9 1132.46    49.8 1116.71    79.7 1099.49
    89.7 1093.29    99.6 1085.27   139.5    1064   159.4 1055.87   169.4 1049.79
   179.4 1045.02   189.3 1043.41   209.3 1042.75     289 1043.51   328.8 1043.14
   338.5 1041.98   348.2 1041.83  361.36 1038.93   367.6 1037.87   377.3 1038.18
   379.2 1039.01     387  1042.3   416.1 1059.92   445.2 1075.25   454.9 1078.38
   464.6 1080.82   551.9 1129.87   571.3 1141.99   581.1 1144.58   600.5 1150.72
#Mann= 3 , 0 , 0
       0     .06       0  361.36    .045       0   379.2      .1       0
Bank Sta=361.36,379.2
XS Rating Curve= 0 ,0
Exp/Cntr=0.3,0.1

Type RM Length L Ch R = 1 ,7507.6  ,228,231.3,234.6
XS GIS Cut Line= 4
     1697080.212      202754.857     1697253.287      202913.306
      1697386.14      203048.597      1697554.34      203191.201
#Sta/Elev= 30
     9.8 1186.42    48.9 1164.57    58.7 1161.01    97.8 1140.74   127.1 1123.44
   136.9 1116.65   146.7 1107.72     176  1088.7   205.3 1072.75   224.9  1066.4
   234.7 1061.26   244.6 1055.86   264.6 1041.61   274.6 1037.69   284.5    1037
   324.5 1039.04   334.4 1038.71   344.4 1035.95   354.4 1034.01   364.4 1034.93
   384.3 1040.13   464.4 1068.65   484.4 1077.24   504.5 1088.85   524.5 1098.45
   544.5 1103.69   574.6  1117.7   594.7  1127.8   604.7 1134.64   644.8 1152.82
#Mann= 3 , 0 , 0
     9.8     .06       0   344.4    .045       0   364.4      .1       0
#XS Ineff= 2 , 0
       0     324                       0
Permanent Ineff=
       F       F
Bank Sta=344.4,364.4
XS Rating Curve= 0 ,0
Exp/Cntr=0.3,0.1

Type RM Length L Ch R = 1 ,7276.3  ,285,287.4,289.9
XS GIS Cut Line= 4
     1696919.325       202887.71     1697131.403      203102.226
     1697216.722       203224.11     1697304.478      203450.814
#Sta/Elev= 30
    10.1 1200.36    50.3 1176.62    70.4 1161.97   100.6 1145.52   120.7 1132.59
   130.7 1129.47   140.8 1125.09   160.9 1112.14   170.9 1104.97     181 1096.08
     191 1089.41   271.5  1039.4   281.5  1034.7   301.7 1032.88   341.3 1033.27
   361.1 1028.21   371.1 1027.16   381.1 1028.67   410.8 1040.68   420.7 1043.68
   430.6 1044.59   440.5 1048.66   541.6 1096.15   551.7 1096.43   592.2 1116.66
   622.6 1129.95   642.9 1140.58     653 1144.65   663.1 1145.99   693.5 1163.03
#Mann= 3 , 0 , 0
       0     .06       0   361.1    .045       0   381.1      .1       0
Bank Sta=361.1,381.1
XS Rating Curve= 0 ,0
Exp/Cntr=0.3,0.1

Type RM Length L Ch R = 1 ,6988.8  ,243.9,236.2,228.5
XS GIS Cut Line= 4
     1696764.533      203002.281     1696875.447      203207.046
     1696969.298      203382.559     1697032.677      203592.199
#Sta/Elev= 30
    10.1 1181.97    30.4 1173.84    60.7 1155.78    70.9 1155.72      81 1149.89
   131.6  1115.6   151.9 1100.09   182.2 1078.53   202.5 1071.91   252.8 1038.51
   262.7    1034   272.7 1031.86   312.5  1027.3   332.4 1026.71  346.32  1024.5
   352.3 1023.33   362.2 1023.13  366.08 1024.88   372.2 1027.69   392.1 1046.22
     402 1053.41     422 1064.88   431.9 1068.71   441.9 1070.18   481.7 1087.98
   541.4 1111.02   561.3 1114.68   581.2 1121.06   601.1 1125.99   650.9 1148.89
#Mann= 3 , 0 , 0
    10.1     .06       0  346.32    .045       0  366.08      .1       0
Bank Sta=346.32,366.08
XS Rating Curve= 0 ,0
Exp/Cntr=0.3,0.1

Type RM Length L Ch R = 1 ,6752.6  ,200.8,204.8,208.7
XS GIS Cut Line= 4
     1696454.948      203294.802     1696679.214      203389.872
     1696791.347      203483.722     1696965.641       203601.95
#Sta/Elev= 30
     9.7 1109.26    19.5 1105.49    48.7 1096.15    77.9 1087.66    97.4 1077.01
   126.7 1063.81   146.2 1056.61   165.6 1050.74   185.1 1040.89   204.6 1033.77
   214.4 1031.58   243.6 1028.03   263.1 1024.91   301.8 1017.59   311.8 1017.11
   321.8 1019.32   341.1 1028.22   360.6 1036.06   370.3 1040.58   389.8 1047.04
   409.9 1056.71     460 1084.94     470 1091.61   480.1 1099.85   510.2 1117.05
   530.2 1127.14   540.2  1130.7   580.4 1141.87   590.4 1146.38   600.4 1146.87
#Mann= 3 , 0 , 0
       0     .06       0   301.8    .045       0   321.8      .1       0
Bank Sta=301.8,321.8
XS Rating Curve= 0 ,0
Exp/Cntr=0.3,0.1

Type RM Length L Ch R = 1 ,6547.8  ,218.7,220.6,222.5
XS GIS Cut Line= 4
     1696385.049      203374.866     1696532.393      203502.708
     1696655.902      203656.553     1696749.075      203823.398
#Sta/Elev= 30
     9.8 1126.25    19.5 1117.13    58.5 1098.31      78 1090.45   107.3 1080.52
     117 1076.55   126.8 1070.75   156.1  1059.1   185.3 1044.89   195.1 1041.12
   224.7 1036.09   234.5 1032.13   254.3 1022.47   264.1 1019.53   283.9 1015.01
   293.6 1013.54   303.6 1012.24   313.6 1012.61   323.3 1016.92     343  1036.2
   352.9 1043.64   372.6 1059.99   382.5 1065.41   392.4 1071.91   402.4 1077.04
   412.5 1079.35   492.9 1125.91   543.2 1151.05   553.3 1158.39   583.5 1175.95
#Mann= 3 , 0 , 0
       0     .06       0   293.6    .045       0   313.6      .1       0
Bank Sta=293.6,313.6
XS Rating Curve= 0 ,0
Exp/Cntr=0.3,0.1

Type RM Length L Ch R = 1 ,6327.2  ,272.5,263,253.6
XS GIS Cut Line= 4
     1696166.083      203494.692     1696391.568      203667.767
     1696470.793      203788.432     1696631.679      203923.723
#Sta/Elev= 30
     9.8 1149.67    39.2 1133.71      49 1130.36    58.8 1128.93    68.6 1124.93
      98 1110.96   117.6 1100.56   127.4 1096.03   205.8 1061.99   225.4 1052.79
     245 1049.96   284.3 1033.71   322.7 1015.47   332.4 1011.47   341.6 1010.04
   351.6 1008.98   361.6 1011.56   370.9 1017.14   380.5 1021.96   390.1 1024.61
     419 1042.32   468.6 1068.32   478.6 1075.55   498.7 1085.94   528.7 1100.52
   538.7 1104.51   548.7 1109.87   568.7 1115.33   608.8 1140.91   638.8 1161.09
#Mann= 3 , 0 , 0
       0     .06       0   341.6    .045       0   361.6      .1       0
Bank Sta=341.6,361.6
XS Rating Curve= 0 ,0
Exp/Cntr=0.3,0.1

Type RM Length L Ch R = 1 ,6064.2  ,190.7,188.8,186.9
XS GIS Cut Line= 4
     1695995.446      203662.892     1696129.518      203793.307
     1696264.809      203871.313      1696463.48      204017.574
#Sta/Elev= 30
     9.8  1090.7    29.5 1081.92    68.9 1067.57    78.8 1065.98    88.6 1065.74
   137.8 1050.97   157.5 1044.62   167.4 1041.12     187 1032.21   226.1 1018.18
   255.4 1005.75   264.9 1003.78   274.9 1003.06   284.9 1004.21   313.9 1007.41
   323.7 1008.89   333.4 1011.68   353.1 1019.37   362.9 1024.16   372.8  1029.7
   392.5 1037.72   451.8 1064.15   461.6 1068.99   471.5 1075.88   491.2 1081.55
   550.4 1108.63   560.3 1113.28   570.2 1120.47     580 1125.68   589.9 1130.32
#Mann= 3 , 0 , 0
       0      .1       0   264.9    .045       0   284.9      .1       0
Bank Sta=264.9,284.9
XS Rating Curve= 0 ,0
Exp/Cntr=0.3,0.1

Type RM Length L Ch R = 1 ,5875.4  ,185.9,206.2,226.4
XS GIS Cut Line= 4
     1695867.468      203795.745     1696047.856       203968.82
     1696208.742       204041.95     1696385.474      204095.579
#Sta/Elev= 30
      10 1061.87      30 1055.62      50  1050.4     100  1038.6     150 1028.04
     160 1025.68     170  1025.1     190 1022.01     220  1016.2     230 1014.83
   259.8 1012.48   269.6 1010.85   279.4 1008.57   289.3 1004.89   298.9 1000.83
   308.9   998.8   318.9  999.51   348.2 1007.31     358 1014.19   387.4 1029.91
   407.1 1038.82   416.9 1044.61   436.4 1051.91   446.2 1058.04   504.5 1081.41
   523.9 1091.38   562.8 1106.34     592  1117.1   601.7 1122.58   611.4 1126.63
#Mann= 3 , 0 , 0
       0      .1       0   298.9    .045       0   318.9     .08       0
Bank Sta=298.9,318.9
XS Rating Curve= 0 ,0
Exp/Cntr=0.3,0.1

Type RM Length L Ch R = 1 ,5669.2  ,230.7,208.5,186.3
XS GIS Cut Line= 4
     1695845.529      203809.152     1695927.191      204034.637
     1695945.473       204157.74     1696108.798      204311.313
#Sta/Elev= 30
      10 1060.44      30 1051.57      40 1048.16    69.9 1039.01    89.9 1033.52
   109.9 1030.95   149.9 1021.84   209.8 1009.73   219.8 1009.32   229.8 1007.85
     259 1001.42   277.7  996.62   287.7  994.75   297.7   994.9   316.4  999.36
     326  999.51   345.1  1002.4   354.7 1005.84   383.8 1018.57   422.8 1036.62
   442.2    1046     452 1052.47   461.7  1057.3   471.5 1059.54   510.5 1080.52
   539.7 1097.69   549.5 1104.03   559.2 1111.78     569 1121.42   588.5 1134.34
#Mann= 3 , 0 , 0
       0      .1       0   277.7    .045       0   297.7      .1       0
Bank Sta=277.7,297.7
XS Rating Curve= 0 ,0
Exp/Cntr=0.3,0.1

Type RM Length L Ch R = 1 ,5460.7  ,217.5,211.7,205.9
XS GIS Cut Line= 4
      1695498.16      204134.582     1695751.678      204201.618
     1695889.407      204249.153     1696084.421      204313.751
#Sta/Elev= 30
    10.1 1106.98    40.3 1092.01    50.4 1082.27   110.9 1050.48   131.1 1036.83
   141.2 1030.65   161.4 1021.42   181.5 1013.12   191.6 1009.31   211.8  999.86
     232  994.92   242.1  993.28   252.1  992.24   281.7  991.09   300.8  989.51
   310.8  989.19   320.8  989.95   330.2   991.7   349.7  996.04   369.1  999.15
   398.2 1010.82   437.3 1027.52   456.8 1038.79   466.6 1043.58     496 1055.71
   525.3 1068.23   535.1 1075.08   544.9 1081.13   564.5 1091.63   613.4  1119.8
#Mann= 3 , 0 , 0
       0      .1       0   300.8    .045       0   320.8      .1       0
Bank Sta=300.8,320.8
XS Rating Curve= 0 ,0
Exp/Cntr=0.3,0.1

Type RM Length L Ch R = 1 ,5249    ,161.4,165.3,169.3
XS GIS Cut Line= 4
     1695426.248      204329.596     1695599.323      204360.067
     1695782.149      204369.818      1696001.54      204444.167
#Sta/Elev= 30
     9.8 1114.14    29.3 1098.15    48.8 1083.12    58.6 1071.56    68.3 1063.73
    97.6    1048   126.9 1033.84   136.7 1028.14   146.4 1020.84     166 1013.16
   204.6  1000.1   214.3  993.23   223.9  988.55   233.6  984.49   242.8   982.3
   252.8  981.83   262.8  982.82   281.7     986     301  990.15   358.8  997.38
   368.9   999.1     379  1002.2   439.4 1031.17   459.5 1045.47   489.8 1062.92
     520 1080.98     530 1087.49   540.1 1096.86   560.3 1106.71   590.5 1124.36
#Mann= 3 , 0 , 0
       0      .1       0   242.8    .045       0   262.8      .1       0
Bank Sta=242.8,262.8
XS Rating Curve= 0 ,0
Exp/Cntr=0.3,0.1

Type RM Length L Ch R = 1 ,5083.7  ,236,236.7,237.4
XS GIS Cut Line= 4
     1695411.622      204468.544      1695571.29      204506.328
     1695749.241      204551.425     1695978.382      204619.679
#Sta/Elev= 30
     9.7 1098.19    19.3 1090.38    38.6 1079.15    77.2 1057.94    86.9 1048.06
    96.5 1042.95   125.5 1030.19   154.4 1016.64   164.1 1010.87   173.7 1003.56
   193.1  994.56   212.4  984.25   221.7  980.11   231.7   978.4   241.7  979.47
     251  984.75   260.7  989.38   289.7  998.44     309 1001.72   318.7 1004.76
   328.3 1010.87   397.5  1035.7   417.4  1049.8   457.2 1071.03   487.1 1088.08
   497.1 1098.58   556.9 1131.88   566.8 1140.76   576.8 1148.12   586.7 1153.65
#Mann= 3 , 0 , 0
       0      .1       0   221.7    .045       0   241.7      .1       0
Bank Sta=221.7,241.7
XS Rating Curve= 0 ,0
Exp/Cntr=0.3,0.1

Type RM Length L Ch R = 1 ,4847    ,207.4,210.7,214.1
XS GIS Cut Line= 4
     1695357.994      204708.655     1695528.631      204733.032
     1695693.174      204780.566      1695896.72      204803.724
#Sta/Elev= 30
     9.6 1090.46    47.9 1068.73    76.6 1051.73    86.2 1042.28    95.8 1036.18
   143.6 1015.13   153.2  1009.8   162.8 1002.57   182.4  994.72   212.7  983.51
   232.9  975.34   242.9   972.8   252.9   975.6   273.1   989.1   283.2  993.02
   293.3  994.56   303.3  995.66   313.4  997.15   323.5  999.86   343.6 1007.44
   382.7 1024.35   392.4  1029.3   402.2 1037.53   441.2 1056.94   470.5  1072.2
   480.2 1081.89     490 1088.88   499.7 1094.49   538.7 1116.13   548.5 1122.69
#Mann= 3 , 0 , 0
       0      .1       0   232.9    .045       0   252.9      .1       0
Bank Sta=232.9,252.9
XS Rating Curve= 0 ,0
Exp/Cntr=0.3,0.1

Type RM Length L Ch R = 1 ,4636.3  ,243.9,245,246
XS GIS Cut Line= 4
     1695314.115      204863.447     1695464.033      204918.295
     1695595.667      204981.675     1695824.809      204996.301
#Sta/Elev= 30
      10 1094.84    29.9  1081.8    49.9 1069.87    69.8 1054.69    79.8 1046.65
    99.8 1036.73   139.7  1019.8   149.7 1012.17   159.6 1007.34   188.9  994.55
   218.1  980.94   227.8  975.36   237.3  969.37   247.3  968.12   257.3   970.6
   266.8  973.08   276.5  974.26     296  975.25   315.7  976.79   325.7  978.44
   335.7  980.73   345.7  984.39   385.6 1003.77   395.6 1009.86   405.6 1017.21
   415.5 1023.53   435.5 1033.83   465.5 1050.69   485.4 1067.66   535.3 1096.19
#Mann= 3 , 0 , 0
       0      .1       0   237.3    .045       0   257.3      .1       0
Bank Sta=237.3,257.3
XS Rating Curve= 0 ,0
Exp/Cntr=0.3,0.1

Type RM Length L Ch R = 1 ,4391.3  ,291.6,296.1,300.7
XS GIS Cut Line= 4
      1695225.14      204993.863     1695371.401      205141.342
     1695482.315      205202.284     1695862.592      205108.434
#Sta/Elev= 30
     9.9  1119.7    19.8 1114.28    29.7 1107.43    59.3 1093.17      89 1076.01
   128.6 1048.76   138.5 1037.78   158.3 1027.36   227.2  985.13   236.9  978.23
   246.6  966.51   256.1  961.92   266.1  960.93   276.1  962.45   295.3  967.02
   344.3  967.21   384.5  968.34     505  974.87     515  976.37   525.1  980.08
   555.2  996.84   565.3 1006.44   575.3 1013.92   585.3 1019.71   605.4 1030.22
   625.5 1037.02   635.6 1043.28   645.6  1050.4   715.9 1086.63   725.9 1094.44
#Mann= 3 , 0 , 0
       0      .1       0   256.1    .045       0   276.1      .1       0
Bank Sta=256.1,276.1
XS Rating Curve= 0 ,0
Exp/Cntr=0.3,0.1

Type RM Length L Ch R = 1 ,4095.2  ,325.2,336.9,348.7
XS GIS Cut Line= 4
     1695127.633      205087.713     1695214.171      205371.703
     1695332.398      205476.523     1695527.412      205784.889
#Sta/Elev= 30
     9.9 1126.03    89.1 1070.09      99 1068.89   108.9 1062.66   158.3 1026.61
     188 1006.38   207.8  995.98   217.7  994.98   257.3  976.53   277.1   969.3
   296.9  963.69   316.6  961.76   336.4  961.69   365.9  956.97   375.9  955.49
   385.9  956.83   454.9  983.45   485.3  997.77   495.4 1003.43   505.6 1005.16
   556.2 1031.11   606.9 1060.69     617 1064.35   627.2 1066.65   647.4 1078.52
     688 1106.37   738.7 1142.39   748.8 1146.94   758.9 1149.61   819.7 1192.17
#Mann= 3 , 0 , 0
       0      .1       0   365.9    .045       0   385.9      .1       0
Bank Sta=365.9,385.9
XS Rating Curve= 0 ,0
Exp/Cntr=0.3,0.1

Type RM Length L Ch R = 1 ,3758.2  ,276.9,276.3,275.6
XS GIS Cut Line= 4
     1694882.647      205215.691     1694948.464      205432.645
     1694995.999      205604.501     1695100.819      205895.803
#Sta/Elev= 30
     9.9 1076.31    19.7 1067.77    39.4 1053.16    49.3 1051.74    98.6 1023.02
   147.9  999.59   157.7  999.27   197.1  982.74   256.4  964.49   296.1  956.38
     306  955.27   325.7  950.01   335.7  949.09   345.7  950.83   365.4  956.11
   385.2  958.09     415   963.4     425  966.31     435  971.98     455  987.56
   464.9   992.3   484.9  997.35   534.9 1003.02   564.8 1009.55   594.8 1019.69
   604.8 1021.39   624.7  1027.9   654.7  1040.9   704.6 1059.25   714.6 1061.84
#Mann= 3 , 0 , 0
       0      .1       0   325.7    .045       0   345.7      .1       0
Bank Sta=325.7,345.7
XS Rating Curve= 0 ,0
Exp/Cntr=0.3,0.1

Type RM Length L Ch R = 1 ,3482    ,352.8,354.1,355.3
XS GIS Cut Line= 4
     1694618.159      205316.855     1694696.164      205538.683
     1694766.857      205764.169     1694818.048      206055.471
#Sta/Elev= 30
     9.8 1058.46    19.6 1053.92    29.4 1053.32    39.2 1049.47   127.4  1007.6
   137.2 1006.71   205.8  974.59     245  965.32   254.8  965.02   353.3  947.14
   363.1  946.67   372.8  944.24   382.8  943.72   392.8  944.67   422.2  951.15
   432.1  955.58   461.6  978.77   471.5  983.85   481.3  985.25     501  994.93
   550.3 1022.42     570 1034.45   579.9 1035.83   589.8 1040.92   639.1 1073.84
   668.6 1095.98   678.5 1100.82   688.3 1103.56   727.8 1133.99   767.2 1167.49
#Mann= 3 , 0 , 0
       0      .1       0   372.8    .045       0   392.8      .1       0
Bank Sta=372.8,392.8
XS Rating Curve= 0 ,0
Exp/Cntr=0.3,0.1

Type RM Length L Ch R = 1 ,3127.9  ,250,248,246
XS GIS Cut Line= 4
      1694270.79      205449.708      1694375.61      205654.473
     1694426.801      205866.551     1694409.737      206206.607
#Sta/Elev= 30
      10 1033.41      60 1020.92      80 1018.54     140 1000.45     190  979.16
     200  978.31     220  971.31   259.8  952.05   269.7  948.32     349  941.04
     359  940.87     369  943.58   398.6  956.52   408.5  959.94   428.4  963.14
   438.3  968.53   458.2  984.97   478.2  997.89   508.3  1014.1   518.3 1018.18
   528.3 1019.61   538.3  1025.8   558.4 1040.87   588.4 1066.84   608.4 1080.39
   618.4 1085.84   628.5 1086.58   718.6  1145.1   728.6 1145.44   788.7 1180.88
#Mann= 3 , 0 , 0
       0     .08       0     349    .045       0     369      .1       0
Bank Sta=349,369
XS Rating Curve= 0 ,0
Exp/Cntr=0.3,0.1

Type RM Length L Ch R = 1 ,2879.9  ,133.4,133.8,134.1
XS GIS Cut Line= 4
     1694087.964      205608.157     1694142.812      205772.701
     1694190.346      205907.991     1694350.014      206205.388
#Sta/Elev= 30
     9.6  969.25    38.5  968.93    86.7  970.59   125.3  969.94   134.9  966.63
   144.5  959.71   154.2   951.6   163.8  945.19   173.4  942.55   221.2  940.43
   230.8  939.65   239.9  938.05   249.9  936.53   259.9  938.26   278.6  948.69
   316.8  968.35   326.8   971.6   336.7  972.97   366.5  987.44   396.3 1004.31
     436 1030.11   445.9 1033.33   455.8 1040.32   465.8 1046.36   525.3 1092.41
     565 1121.95     575    1123   584.9 1129.31   634.5 1163.62   654.4 1178.06
#Mann= 3 , 0 , 0
       0     .08       0   239.9    .045       0   259.9      .1       0
Bank Sta=239.9,259.9
XS Rating Curve= 0 ,0
Exp/Cntr=0.3,0.1

Type RM Length L Ch R = 1 ,2746.2  ,246.7,240.7,234.7
XS GIS Cut Line= 4
     1693885.618      205681.653     1694023.347      205830.351
     1694069.663       205968.08     1694178.139      206196.002
#Sta/Elev= 30
    10.1  997.77    20.3  996.06    40.5  991.03    81.1   978.6   131.7  968.31
   141.9  963.86     152  957.03   162.1  954.93   172.3  945.93   182.4  939.91
   192.5  939.02   241.4  937.92   251.1  937.28   260.5  935.47   270.5  933.68
   280.5  933.88   289.9  935.31   309.2  946.88   318.9  951.88   378.3  978.45
   388.4  982.62   398.5  984.13   408.6  987.72   418.7  992.81   438.9 1007.77
   489.3 1038.98   509.5 1052.27   519.6 1055.26   529.7 1060.17   600.4  1107.7
#Mann= 3 , 0 , 0
       0     .08       0   260.5    .045       0   280.5      .1       0
Bank Sta=260.5,280.5
XS Rating Curve= 0 ,0
Exp/Cntr=0.3,0.1

Type RM Length L Ch R = 1 ,2505.5  ,404.7,407.4,410
XS GIS Cut Line= 4
     1693602.867      205750.762     1693773.504      205925.055
     1693894.169      206094.474     1694094.058      206358.962
#Sta/Elev= 30
     9.8 1088.54    19.5 1080.34    29.3  1070.1    48.8 1052.73    87.8 1024.03
   136.6  991.19   156.1  974.65   293.4  938.74   303.3  936.53     343  931.44
   352.8  928.65   362.8  927.07   372.8  927.49   382.6  929.49   402.4  935.91
   432.1  954.35     442  957.62   451.9  958.56     472  964.21   512.2  976.61
   532.3   985.1   552.4  996.33   572.5 1012.11   582.5 1017.92   592.6 1020.22
   632.7 1044.36   703.1 1082.02   723.2 1096.93   733.2 1099.52   783.4 1128.44
#Mann= 3 , 0 , 0
       0     .08       0   352.8    .045       0   372.8      .1       0
Bank Sta=352.8,372.8
XS Rating Curve= 0 ,0
Exp/Cntr=0.3,0.1

Type RM Length L Ch R = 1 ,2098.2  ,349.3,348.5,347.7
XS GIS Cut Line= 4
     1693323.753      205982.341     1693448.074      206146.884
     1693527.299      206296.801     1693693.061      206488.159
#Sta/Elev= 30
     9.8 1028.29    19.6 1021.08    29.5 1015.23    58.9  999.97    78.6  990.83
    88.4  989.62    98.2  986.46   157.1  960.06   176.8  949.07   206.2  939.08
   216.2  937.63   256.1  928.89     286  923.62     296  919.92     306  918.57
     316  921.57   325.9  929.81   335.9  935.23   345.9  938.77   355.8  946.88
   365.8  954.03   416.3  985.48   466.9  1014.9   477.1 1019.32   487.2 1022.89
   547.9 1061.34   598.6  1092.8   608.7 1100.23   618.8 1106.42     629 1110.05
#Mann= 3 , 0 , 0
       0      .1       0     296    .045       0     316      .1       0
Bank Sta=296,316
XS Rating Curve= 0 ,0
Exp/Cntr=0.3,0.1

Type RM Length L Ch R = 1 ,1749.7  ,221.7,218.7,215.7
XS GIS Cut Line= 4
     1693003.198      206126.164     1693123.863      206288.269
     1693218.933      206451.593     1693317.658      206661.233
#Sta/Elev= 30
    10.1 1051.98    30.3 1039.61    60.6 1019.78    70.7 1012.72    80.8  1004.3
    90.9  997.41   111.1  986.16   131.4  980.28   171.8   961.7   231.9  936.64
   251.8  930.14   261.8   929.2   281.7  922.15   311.4  915.65   321.4  914.85
   331.4  916.92   351.3  928.85   371.2   939.3   381.1  943.45   391.1  945.55
   411.2  958.03   491.8 1001.34   501.9 1002.31   532.1 1019.53   552.3 1028.33
   572.4 1038.12   592.6 1050.31   602.6  1057.8   612.7 1067.07   622.8  1067.7
#Mann= 3 , 0 , 0
       0     .08       0   311.4    .045       0   331.4      .1       0
Bank Sta=311.4,331.4
XS Rating Curve= 0 ,0
Exp/Cntr=0.3,0.1

Type RM Length L Ch R = 1 ,1531    ,150.9,153.5,156.1
XS GIS Cut Line= 4
     1692876.759      206198.914      1692959.64      206456.089
     1693025.457      206537.751     1693142.466      206763.236
#Sta/Elev= 30
      10 1080.57      40 1062.84      50 1056.17    80.1 1033.34   110.1 1008.24
   120.1 1003.73   130.1 1000.65   180.1  962.09   200.1  948.53   210.2  942.68
   220.2  937.22   230.2  936.28   270.2  920.52   279.7  918.64   307.9  915.31
   317.9  913.17   327.9  914.01   346.5  926.28     356  931.18   365.5  932.69
   375.1  937.04   433.7  969.26   482.6  997.66   492.3  998.76   502.1 1003.56
   531.4 1022.97     551 1033.62   609.6  1062.7   619.3 1063.71   629.1  1068.8
#Mann= 3 , 0 , 0
       0     .08       0   307.9    .045       0   327.9      .1       0
Bank Sta=307.9,327.9
XS Rating Curve= 0 ,0
Exp/Cntr=0.3,0.1

Type RM Length L Ch R = 1 ,1377.5  ,258,261.5,265
XS GIS Cut Line= 4
     1692711.778      206293.742     1692780.032       206442.44
     1692915.324      206664.269     1692995.767      206859.283
#Sta/Elev= 30
     9.6 1069.89    38.5 1049.27   105.9   993.3   115.5  986.73   125.1  982.84
   134.7  974.14     154  947.22   163.6  935.25   173.6  926.65   183.6  920.82
   203.6  914.47   223.6  910.92   253.6  910.44   293.5  913.09   313.5  911.76
   323.5     910   333.5  910.23   343.5  914.48   363.5  929.39   373.5  931.08
   383.5   936.3   463.6  985.49   483.7  999.95   493.8 1004.88   503.8 1007.68
   533.9 1028.21   594.2 1064.29   604.3 1067.51   624.4 1077.19   634.4 1083.83
#Mann= 3 , 0 , 0
       0     .08       0   313.5    .045       0   333.5      .1       0
Bank Sta=313.5,333.5
XS Rating Curve= 0 ,0
Exp/Cntr=0.3,0.1
